--- HNGRDCK_1.prj (project) ---

Proj Title=HNGRDCK_1
Current Plan=p01
Default Exp/Contr=0,0
English Units
Geom File=g01
Flow File=f01
Plan File=p01
BEGIN DESCRIPTION:
Stream Name: Hungard Creek
Flood Zone: Approximate
Summers County, West Virginia
HEC-RAS Version: 5.0.7
Hydrology Method:
Regression.
Model Notes:
END DESCRIPTION:
DSS File=dss
DSS Export Rating Curves= 0
DSS Export Rating Curve Sorted= 0
DSS Export Volume Flow Curves= 0
DXF Filename=HNGRDCK_A.
DXF OffsetX= 0
DXF OffsetY= 0
DXF ScaleX= 0
DXF ScaleY= 0

--- HNGRDCK_1.p01 (plan) ---

Plan Title=Floodplain
Program Version=5.07
Short Identifier=Floodplain
Geom File=g01
Flow File=f01
Subcritical Flow
K Sum by GR= 0
Std Step Tol= 0.01
Critical Tol= 0.01
Num of Std Step Trials= 20
Max Error Tol= 0.3
Flow Tol Ratio= 0.001
Split Flow NTrial= 30
Split Flow Tol= 0.02
Split Flow Ratio= 0.02
Log Output Level= 0
Friction Slope Method= 1
Unsteady Friction Slope Method= 2
Unsteady Bridges Friction Slope Method= 1
Parabolic Critical Depth
Global Vel Dist= 0 , 0 , 0
Global Log Level= 0
CheckData=True
Encroach Param=-1 ,0,0, 0
Computation Interval=0.1SEC
Output Interval=1MIN
Instantaneous Interval=Max Profile
Mapping Interval=1HOUR
Computation Time Step Use Courant=        0
Computation Time Step Use Time Series=    0
Computation Time Step Count To Double=0
Computation Time Step Max Doubling=0
Computation Time Step Max Halving=0
Computation Time Step Residence Courant=0
Run HTab= 0
Run UNet= 0
Run Sediment= 0
Run PostProcess= 0
Run WQNet= 0
Run RASMapper= 0
UNET Theta= 0
UNET Theta Warmup= 0
UNET ZTol= 0
UNET ZSATol= 0
UNET MxIter= 0
UNET Max Iter WO Improvement= 0
UNET MaxInSteps= 0
UNET DtIC= 0
UNET DtMin= 0
UNET MaxCRTS= 0
UNET WFStab= 0
UNET SFStab= 0
UNET WFX= 1
UNET SFX= 1
UNET 1D Methodology=Finite Difference
UNET DSS MLevel= 1
UNET Pardiso=0
UNET DZMax Abort= 0
UNET Use Existing IB Tables= 0
UNET Froude Reduction=False
UNET Froude Limit= 0
UNET Froude Power= 0
UNET D1 Cores= 0
UNET D2 Coriolis=0
UNET D2 Cores= 0
UNET D2 Theta= 1
UNET D2 Theta Warmup= 1
UNET D2 Z Tol= 0.01
UNET D2 Volume Tol= 0.01
UNET D2 Max Iterations= 20
UNET D2 Equation= 0
UNET D2 RampUpFraction=0.1
UNET D2 TimeSlices= 1
UNET D2 BCVolumeCheck=0
UNET D1D2 MaxIter= 0
UNET D1D2 ZTol=0.01
UNET D1D2 QTol=0.1
UNET D1D2 MinQTol=1
DSS File=dss
Write IC File= 0
Write IC File at Fixed DateTime=0
Write IC File at Sim End=0
Echo Input=False
Echo Parameters=False
Echo Output=False
Write Detailed= 0
HDF Write Warmup=0
HDF Write Time Slices=0
HDF Flush=0
HDF Face Node Velocities=0
HDF Compression= 1
HDF Chunk Size= 1
HDF Spatial Parts= 1
HDF Use Max Rows=0
HDF Fixed Rows= 1
Calibration Method= 0
Calibration Iterations= 20
Calibration Max Change=0.05
Calibration Tolerance=0.2
Calibration Maximum=1.5
Calibration Minimum=0.5
Calibration Optimization Method= 1
WQ AD Non Conservative
WQ ULTIMATE=-1
WQ Max Comp Step=1HOUR
WQ Output Interval=15MIN
WQ Output Selected Increments= 0
WQ Output face flow=0
WQ Output face velocity=0
WQ Output face area=0
WQ Output face dispersion=0
WQ Output cell volume=0
WQ Output cell surface area=0
WQ Output cell continuity=0
WQ Output cumulative cell continuity=0
WQ Output face conc=0
WQ Output face dconc_dx=0
WQ Output face courant=0
WQ Output face peclet=0
WQ Output face adv mass=0
WQ Output face disp mass=0
WQ Output cell mass=0
WQ Output cell source sink temp=0
WQ Output nsm pathways=0
WQ Output nsm derived pathways=0
WQ Output MaxMinRange=-1
WQ Daily Max Min Mean=-1
WQ Daily Range=0
WQ Daily Time=0
WQ Create Restart=0
WQ Fixed Restart=0
WQ System Summary=0
WQ Write To DSS=0
WQ Use Fixed Temperature=0
Sorting and Armoring Iterations= 10
XS Update Threshold= 0.02
Bed Roughness Predictor= 0
Hydraulics Update Threshold= 0.02
Energy Slope Method= 1
Volume Change Method= 1
Sediment Retention Method= 0
XS Weighting Method= 0
Number of US Weighted Cross Sections= 1
Number of DS Weighted Cross Sections= 1
Upstream XS Weight=0
Main XS Weight=1
Downstream XS Weight=0
Number of DS XS's Weighted with US Boundary= 1
Upstream Boundary Weight= 1
Weight of XSs Associated with US Boundary= 0
Number of US XS's Weighted with DS Boundary= 1
Downstream Boundary Weight= 0.5
Weight of XSs Associated with DS Boundary= 0.5
Percentile Method= 0
Sediment Output Level= 3
Mass or Volume Output= 0
Output Increment Type= 1
Profile and TS Output Increment= 1
XS Output Flag= 0
XS Output Increment= 10
Write Gradation File= 0
Read Gradation Hotstart= 0
Write HDF5 File= 1
Write Binary Output= 1
Write DSS Sediment File= 0
SV Curve= 0
Specific Gage Flag= 0

--- HNGRDCK_1.f01 (steady flow) ---

Flow Title=Flows
Program Version=5.07
Number of Profiles= 6
Profile Names=01pct,10pct,04pct,02pct,0_2pct,01plus
River Rch & RM=HNGRDCK_1,Main            ,17282
    2086    1159    1505    1786    2845    3086
River Rch & RM=HNGRDCK_1,Main            ,11257
    2344    1308    1694    2009    3189    3466
River Rch & RM=HNGRDCK_1,Main            ,2
    3054    1722    2219    2624    4134    4517
Boundary for River Rch & Prof#=HNGRDCK_1,Main            , 1
Up Type= 0
Dn Type= 1
Dn Known WS=1541.2
Boundary for River Rch & Prof#=HNGRDCK_1,Main            , 2
Up Type= 0
Dn Type= 1
Dn Known WS=1540.4
Boundary for River Rch & Prof#=HNGRDCK_1,Main            , 3
Up Type= 0
Dn Type= 1
Dn Known WS=1540.8
Boundary for River Rch & Prof#=HNGRDCK_1,Main            , 4
Up Type= 0
Dn Type= 1
Dn Known WS=1541
Boundary for River Rch & Prof#=HNGRDCK_1,Main            , 5
Up Type= 0
Dn Type= 1
Dn Known WS=1541.7
Boundary for River Rch & Prof#=HNGRDCK_1,Main            , 6
Up Type= 0
Dn Type= 1
Dn Known WS=1541.8
DSS Import GetInterval= 0
DSS Import GetPeak= 0
DSS Import FillOption= 0

--- HNGRDCK_1.g01 (geometry) ---

Geom Title=Geometry
Program Version=5.07

River Reach=HNGRDCK_1       ,Main
Reach XY= 30
2045402.17700002252605.4460000122045585.51900004252111.260999996
     2045476.789251062.4220000342045116.62300002250338.051000037
     2044475.815250128.868000011     2044536.697249272.988000028
     2044268.045249201.6020000212043763.46400004249307.865000037
2043086.38100002249667.023000036     2042947.492249587.813000015
     2042373.521249845.7420000162041665.71700003249482.921999993
2040908.98299999250004.8530000522040679.82700001249933.314000012
     2040215.417249142.5149999952039787.87600004 248828.25600001
2039890.88399999248293.9860000372040232.32299999247822.248999973
     2040907.257247597.3760000342041111.25000001246516.647000048
2041500.31300002246148.069999982     2041506.563245832.098000002
2041403.09100002245677.9319999632041182.62700001245679.883999975
2041164.89600001245275.847999998      2040607.49244825.057000022
     2040539.829244527.174000022     2039946.195244266.158000008
     2039486.424244224.4590000252039401.01026427243936.116604297

Type RM Length L Ch R = 1 ,17282   ,259,230.7,214.3
XS GIS Cut Line= 4
2045753.79288326253103.4690339342045463.35894855252689.116620413
2045399.46348291252470.323056264 2045306.5246238252342.532124991
#Sta/Elev= 30
       0 1755.83     169 1736.48   238.5 1729.33   261.3 1728.85   265.6 1727.87
   272.8 1724.26   284.4 1724.72     308 1723.98   340.9 1720.58   415.7 1712.58
   468.8 1696.35   508.5 1694.81   531.7 1695.16   573.4 1694.22   580.2 1693.67
   587.1 1691.86   590.5 1691.15     611  1690.7   619.5 1691.66   641.8 1695.36
     676  1696.4   706.7 1695.92   717.4 1693.68   730.6 1692.35   734.1 1692.73
   743.5 1690.47   766.5 1691.58   788.2 1691.47   811.2 1698.06891.9495 1705.56
#Mann= 6 ,-1 , 0
       0    .035       0     169     .04       0   340.9      .1       0
   587.1    .045       0   619.5      .1       0     676     .08       0
#XS Ineff= 2 , 0
                          687.68         1697.55
Permanent Ineff=
       F       F
Bank Sta=587.1,619.5
XS Rating Curve= 0 ,0
Exp/Cntr(USF)=0,0
Exp/Cntr=0.3,0.1

Type RM Length L Ch R = 1 ,17051   ,267.6,262.2,257.8
XS GIS Cut Line= 4
2045951.28795886252557.4532366772045622.12949952252419.981174247
2045436.25178131252342.5321249912045327.82311235252311.552505289
#Sta/Elev= 30
       0 1767.55    88.6 1752.68    99.3 1749.55   111.6 1747.62   209.5 1732.43
   227.3 1730.43   304.7 1726.44   316.1 1721.65     320 1722.13     341 1722.06
     395 1709.43   419.2 1705.46   427.7 1703.07   433.4 1700.63   440.6 1690.07
  444.031686.808   447.7  1685.7  473.671686.809   486.8 1689.06   510.5 1690.41
   525.5 1690.48   535.5 1688.59   547.2 1688.51   557.8 1689.45   561.3 1691.28
   595.3 1690.57     609 1694.24   622.7 1695.18     650 1700.36670.8476 1702.93
#Mann= 6 ,-1 , 0
       0      .1       0   111.6    .035       0     320     .06       0
   427.7     .08       0  444.03    .045       0  473.67     .08       0
#XS Ineff= 2 , 0
                             500            1698
Permanent Ineff=
       F       F
Bank Sta=444.03,473.67
XS Rating Curve= 0 ,0
Exp/Cntr(USF)=0,0
Exp/Cntr=0.3,0.1

Type RM Length L Ch R = 1 ,16789   ,221.8,219,216.6
XS GIS Cut Line= 4
 2045999.9764973252288.7880998632045667.48772884252144.500521099
2045469.87647967252105.2919399132045298.92706569252075.493418211
#Sta/Elev= 30
       0 1759.68      17 1755.19    52.8  1748.5    92.1  1743.2   106.4 1740.11
   123.4 1737.78   152.9 1735.37   220.9 1726.68   225.6 1725.74   231.6 1722.84
   256.6 1723.71   346.1 1717.17   367.2 1716.96   387.3 1715.11   410.7 1709.58
     414 1703.84   418.7 1693.58   420.7  1690.6  427.831684.039   430.7 1682.82
   450.8 1682.36   462.51684.039   477.6 1688.59   527.7 1690.43   561.2 1690.92
   644.4 1689.47   667.8 1692.79   694.4 1698.78   704.4 1702.47737.4373  1705.2
#Mann= 6 ,-1 , 0
       0     .12       0      50    .035       0     160     .04       0
     270      .1       0  427.83    .045       0   462.5      .1       0
#XS Ineff= 2 , 0
                          527.78         1693.33
Permanent Ineff=
       F       F
Bank Sta=427.83,462.5
XS Rating Curve= 0 ,0
Exp/Cntr(USF)=0,0
Exp/Cntr=0.3,0.1

Type RM Length L Ch R = 1 ,16570   ,228.5,221.7,218
XS GIS Cut Line= 4
2046042.32176498251937.479212437  2045725.516429 251923.36412321
2045483.99156889251898.2706312512045127.97765172251906.112347488
#Sta/Elev= 30
       0 1760.45    51.4 1738.69   100.7 1726.39   145.5 1722.53   222.2 1720.36
   248.5 1718.05   268.2 1714.69   291.2 1715.47   389.9 1713.57   406.5 1712.36
   416.4  1710.3   419.7 1708.53     423  1704.1   429.6 1686.28  435.921682.231
   452.7 1680.76   467.8 1682.23   479.1 1683.21     489 1686.87   498.9 1688.03
   591.1 1688.25   654.4    1686     683 1686.89   729.5 1690.27   742.4 1692.98
   761.7 1699.35   780.9 1701.71   853.6 1705.82   882.6 1709.85916.0448 1717.04
#Mann= 8 ,-1 , 0
       0      .1       0   291.2     .04       0   389.9    .035       0
  435.92    .045       0   467.8    .035       0     683      .1       0
   780.9    .035       0   882.6      .1       0
#XS Ineff= 2 , 0
                             500        1691.952
Permanent Ineff=
       F       F
Bank Sta=435.92,467.8
XS Rating Curve= 0 ,0
Exp/Cntr(USF)=0,0
Exp/Cntr=0.3,0.1

Type RM Length L Ch R = 1 ,16348   ,246.5,244.9,242.8
XS GIS Cut Line= 4
2045930.96939441 251659.882457642045606.32234219251684.975949599
2045336.56730363251716.3428145472045079.35901105 251775.93985795
#Sta/Elev= 30
       0 1767.39   143.9 1732.17   183.4 1723.78   193.2 1717.44   196.5 1716.41
   203.1 1717.92   219.6 1717.54   249.2 1713.36   298.5 1709.78     315 1707.37
   318.3 1706.46   324.9  1701.5   334.8 1691.37   344.7 1684.32  364.281680.667
   387.6 1678.98   397.5 1679.23  403.671680.667   410.7 1686.07   427.3 1687.51
   466.9 1685.19   529.6 1685.68   579.2 1683.78   602.4 1685.46   622.6 1685.32
   682.9 1699.14   784.3 1702.04   800.4 1703.94   814.6 1707.34861.2105 1725.15
#Mann= 8 ,-1 , 0
       0      .1       0     180     .06       0     270      .1       0
  364.28    .045       0  403.67    .035       0  575.62      .1       0
  667.19    .035       0  777.19      .1       0
#XS Ineff= 1 ,-1
  426.89  772.161691.079
Permanent Ineff=
       T
Bank Sta=364.28,403.67
XS Rating Curve= 0 ,0
Exp/Cntr(USF)=0,0
Exp/Cntr=0.3,0.1

Type RM Length L Ch R = 1 ,16103   ,268.5,269.5,270.4
XS GIS Cut Line= 4
2045849.41554555251424.630970524 2045600.0489692251435.609373256
2045251.87676827251496.7747599062044867.63267265251719.479501042
#Sta/Elev= 30
       0 1775.02    78.4 1746.22   107.9 1740.93   124.4 1733.29   137.5 1731.15
   147.3 1727.62   170.3 1726.65     190 1720.36   229.4 1711.04   249.1 1704.17
   275.8 1691.52   289.1  1681.1  315.141678.222   329.1 1677.28  357.041678.223
   365.7 1682.05   379.1 1683.64     529 1681.47   532.3 1681.76   548.9 1689.72
   562.3 1693.96   582.3 1697.26   617.3 1695.95   688.2  1697.4     765 1699.91
   852.4 1703.86   867.6 1705.76   941.4 1708.15  1011.7 1716.08 1047.23 1728.79
#Mann= 7 ,-1 , 0
       0      .1       0      90     .04       0     190      .1       0
  289.61    .035       0  315.14    .045       0  357.04    .035       0
  703.11      .1       0
#XS Ineff= 2 , 0
                          378.36          1688.1
Permanent Ineff=
       F       F
Bank Sta=315.14,357.04
XS Rating Curve= 0 ,0
Exp/Cntr(USF)=0,0
Exp/Cntr=0.3,0.1

Type RM Length L Ch R = 1 ,15834   ,279.6,273.9,267.6
XS GIS Cut Line= 4
2045796.09187513251137.6241562422045568.68210425251172.127707686
2045239.33002229251220.7463483562044811.17231574251307.005226966
#Sta/Elev= 30
       0 1774.11    31.9 1761.94   121.5  1732.2   131.5 1725.24   138.1 1722.73
   151.4 1723.32     168 1721.94   181.2 1715.21   192.4 1712.11   224.4  1708.3
   238.6 1705.23   255.9  1696.4   277.4 1679.82  289.811676.328   297.3 1674.81
   316.6 1674.14   327.2 1674.97  329.42 1676.33   333.8  1679.1   340.4 1680.07
   363.7    1679   532.8 1679.37   550.7 1680.91   582.7 1687.67   615.2 1691.87
   706.6 1695.97   821.3  1705.2   860.5 1711.36   921.6 1724.98 999.694  1747.6
#Mann= 7 ,-1 , 0
       0      .1       0     140     .04       0  240.01      .1       0
  289.81    .045       0  329.42      .1       0  340.01    .035       0
  742.93      .1       0
Bank Sta=289.81,329.42
XS Rating Curve= 0 ,0
Exp/Cntr(USF)=0,0
Exp/Cntr=0.3,0.1

Type RM Length L Ch R = 1 ,15560   ,213.8,216,217.6
XS GIS Cut Line= 4
2045772.56672642250830.2288797442045469.87647967250902.372669126
2045196.98475461251016.861726189  2044806.467286251131.350783252
#Sta/Elev= 30
       0 1772.51    31.9 1760.26    55.5  1753.3   102.7 1736.19     133 1728.13
   146.5 1720.27   157.5 1720.93   176.9  1719.3   207.2 1711.16   217.4  1710.7
   281.4 1701.39   336.4    1692   340.3 1690.79   343.8 1686.96     351  1683.5
  363.921674.595   368.7 1672.67  381.331674.596   407.9 1676.89     567 1676.03
   575.1 1677.29   585.8  1682.1   592.9 1687.73   607.1 1691.88   658.4 1691.56
   726.8 1695.21     867 1707.34   894.3 1711.23   942.2  1721.41014.058 1741.16
#Mann= 9 ,-1 , 0
       0      .1       0     120     .04       0     220      .1       0
  321.17    .035       0  363.92    .045       0  381.33    .035       0
  531.17      .1       0   637.1    .035       0   737.1      .1       0
Bank Sta=363.92,381.33
XS Rating Curve= 0 ,0
Exp/Cntr(USF)=0,0
Exp/Cntr=0.3,0.1

Type RM Length L Ch R = 1 ,15344   ,308.9,300.5,296.1
XS GIS Cut Line= 4
2045707.93119209250589.2934929572045439.01088217250686.104804528
2045051.76563589 250841.002903042044729.06126399251000.203726512
#Sta/Elev= 30
       0 1770.12      27 1759.27    59.1 1749.58    87.3 1738.46   118.1 1728.99
   128.1  1723.5   138.6 1724.16     154 1722.83   166.8 1718.34     285 1694.41
     363 1685.43   376.9 1681.82   388.2 1674.69   398.3 1673.72   405.9 1671.35
   415.8 1671.17   426.4 1669.87   444.4 1671.16   453.8 1674.81     550 1673.73
   562.4 1676.79   578.3  1683.2     603 1688.07     649 1688.28   740.1 1691.93
   797.1 1697.67   884.9 1713.11   929.1 1723.97  1027.5 1751.691062.729 1759.43
#Mann= 9 ,-1 , 0
       0      .1       0     160     .04       0     260      .1       0
   415.8    .045       0   444.4      .1       0  475.82    .035       0
  792.89      .1       0  902.89     .05       0 1012.89      .1       0
Bank Sta=415.8,444.4
XS Rating Curve= 0 ,0
Exp/Cntr(USF)=0,0
Exp/Cntr=0.3,0.1

Type RM Length L Ch R = 1 ,15043   ,231.3,228.5,225.8
XS GIS Cut Line= 4
2045546.57900614250283.8000208912045264.75052135250406.427682213
2045021.64656118250589.2934929572044649.46085226250877.576065189
#Sta/Elev= 30
       0 1757.24    48.5 1740.91   104.7 1724.28   116.5 1716.51     138 1716.35
   142.1 1715.27     152 1710.19   166.6 1705.96   198.8  1698.1   241.7 1689.48
   263.2 1687.62   271.7 1685.73   330.1 1681.45   342.9 1678.87   363.4 1672.24
   375.8  1670.1  379.151668.608     384 1667.53  407.261668.606     425 1671.34
   476.8  1671.3   498.9 1674.67   548.2 1677.17   596.8 1683.32   698.9 1685.53
   742.2  1687.7   800.7 1693.44   845.1 1700.67   887.8  1710.41082.329 1769.43
#Mann= 8 ,-1 , 0
       0      .1       0      90     .04       0     200      .1       0
  379.15    .045       0  407.26      .1       0  557.35    .035       0
  891.55     .05       0 1051.55      .1       0
Bank Sta=379.15,407.26
XS Rating Curve= 0 ,0
Exp/Cntr(USF)=0,0
Exp/Cntr=0.5,0.3

Type RM Length L Ch R = 1 ,14815   ,51.2,52.2,54.9
XS GIS Cut Line= 4
2045410.76480537250095.040417529 2045103.3983354250238.621408824
2044987.22476151 250350.492257752044608.58496515250750.645678908
#Sta/Elev= 30
       0 1733.55    36.8 1719.37    47.7 1712.03    69.4 1712.28   145.4 1693.36
   201.2 1686.29   255.4 1680.39   304.8 1676.94   345.4 1675.49   382.6 1672.54
   394.2 1670.63  401.42 1667.28   405.2 1665.72   410.4 1664.94   423.4 1664.75
     428 1665.21  435.291667.278   441.6 1668.24   454.5 1668.76   523.5 1669.43
   604.8  1672.7     668 1676.72   768.2 1687.09   821.2 1690.93   865.3 1697.34
   897.8 1703.95   925.6 1710.97   975.2 1724.97  1029.4 1742.091051.429 1747.94
#Mann= 13 ,-1 , 0
       0     .06       0      50     .04       0     170      .1       0
     270    .035       0  379.25      .1       0  389.25    .035       0
  401.42    .045       0  435.29    .035       0  530.53     .04       0
  660.53    .035       0  670.53     .04       0  930.53      .1       0
  960.53     .05       0
#XS Ineff= 2 , 0
             385 1674.43     450         1674.43
Permanent Ineff=
       F       F
Bank Sta=401.42,435.29
XS Rating Curve= 0 ,0
Exp/Cntr(USF)=0,0
Exp/Cntr=0.5,0.3

Type RM Length L Ch R = 1 ,14763   ,161,155.7,145.6
XS GIS Cut Line= 4
2045383.07545771250034.2419732872045062.52244829250208.502334114
2044899.01889986250359.0977076682044580.61725292250690.407529486
#Sta/Elev= 30
       0  1735.7    25.1 1724.73    36.3 1715.28    40.1 1713.21    58.6 1713.22
    77.9 1709.85   111.8  1701.2   118.5 1699.02   129.7 1693.49   140.9 1691.02
   163.3 1688.37   196.9 1682.12     230 1678.34   298.7 1675.11   393.6 1672.58
   415.1 1670.34  421.071667.186   427.4 1664.92  468.431667.185   587.1 1671.43
   663.8 1675.91   762.7 1683.47   820.7 1689.73   857.7 1695.08   883.3 1696.06
   899.6 1699.63   930.6 1701.93   944.2  1708.4   990.5 1718.891046.652 1735.59
#Mann= 12 ,-1 , 0
       0      .1       0      20     .04       0     280    .035       0
     360     .04       0  421.07    .045       0  468.43    .035       0
  494.86     .04       0  627.15      .1       0  737.15     .04       0
  767.15     .06       0  867.15     .04       0  907.15     .05       0
#XS Ineff= 2 , 0
             410 1674.43     479         1674.43
Permanent Ineff=
       F       F
Bank Sta=421.07,468.43
XS Rating Curve= 0 ,0
Exp/Cntr(USF)=0,0
Exp/Cntr=0.5,0.3

Type RM Length L Ch R = 1 ,14607   ,400.7,412.7,419
XS GIS Cut Line= 4
 2045267.2454136249788.0173232972044930.34204934250103.622199017
2044800.61489183250289.4999172322044529.54321944250624.467055265
#Sta/Elev= 30
       0 1715.56    15.4 1714.25    32.4 1704.23    60.1 1694.45   113.6  1682.5
   150.2 1677.07   232.9 1673.02   350.4 1671.75   415.5    1669   468.9 1668.73
     483 1667.53   527.8 1668.32     539 1667.62  544.671665.928     547 1665.07
   560.8 1664.76  572.861665.927   685.7 1667.87   720.6 1669.52   762.7 1674.42
   804.7  1681.5   838.9 1688.74     870 1693.11   940.2 1699.35  1023.9 1699.48
  1033.1 1702.35  1041.5 1707.66  1054.4 1713.12  1083.7 1718.381119.219 1726.57
#Mann= 12 ,-1 , 0
       0      .1       0     130     .04       0     140    .035       0
     270      .1       0  541.64     .04       0  544.67    .045       0
  572.86      .1       0  728.31     .04       0  788.31     .06       0
  888.31      .1       0 1038.31     .05       0 1048.31      .1       0
#XS Ineff= 1 ,-1
291.6622  471.961672.249
Permanent Ineff=
       T
Bank Sta=544.67,572.86
XS Rating Curve= 0 ,0
Exp/Cntr(USF)=0,0
Exp/Cntr=0.3,0.1

Type RM Length L Ch R = 1 ,14194   ,293.2,305.5,313.7
XS GIS Cut Line= 4
2045255.62805621249737.6754412812044548.90548175 250093.94106786
2044382.39002585250196.5610581242044237.17305849250308.862179546
#Sta/Elev= 30
       0 1708.68    54.7 1693.77   153.9 1674.92   285.2 1670.11   370.6 1669.94
   484.5 1665.09   553.9 1666.12   616.8 1665.15   638.9 1662.84   654.1 1664.23
   682.9 1661.27   697.6 1663.38   727.3 1662.56   778.6  1664.5   808.7  1662.5
   849.5  1663.8   857.6 1661.53   870.3 1659.78   883.7  1661.6   885.8 1662.78
   897.3 1677.41   901.2 1680.47   928.1 1694.35   943.6 1693.99     959 1703.56
   966.7 1706.51  1031.5 1722.29  1093.7 1729.13  1126.5 1735.241170.614 1750.24
#Mann= 4 ,-1 , 0
       0      .1       0   857.6    .045       0   883.7     .04       0
  987.04      .1       0
#XS Ineff= 1 ,-1
 265.249630.0199 1672.11
Permanent Ineff=
       T
Bank Sta=857.6,883.7
XS Rating Curve= 0 ,0
Exp/Cntr(USF)=0,0
Exp/Cntr=0.3,0.1

Type RM Length L Ch R = 1 ,13889   ,297.1,301.2,302.3
XS GIS Cut Line= 5
2045259.50050868249706.6958215782044606.99226869249826.741847925
2044355.28285861249842.2316577772044226.28535059249857.864544282
2044015.05284335250076.468665634
#Sta/Elev= 30
       01703.817    83.6 1688.38  173.671675.242 212.3911672.448 433.8691664.263
  547.291664.401 637.8391660.942 667.3251662.481  683.761659.884 713.3431659.375
 759.3621661.828  769.861658.612 779.0841657.795 802.0931658.633 808.6671659.756
 821.0911657.858 828.3891659.199 831.6761660.314 838.251 1666.87 848.1121672.821
 886.1171683.911 963.4151690.3341064.9511691.5951084.0011695.9431112.3291697.217
1126.4941700.931 1148.561701.3841178.7231705.6311279.3761727.2071349.5711737.129
#Mann= 5 ,-1 , 0
       0      .1       0  769.86    .045       0 802.093      .1       0
  995.64     .04       0 1105.59      .1       0
#XS Ineff= 2 , 0
           663.1 1666.59
Permanent Ineff=
       F       F
Bank Sta=769.86,802.093
XS Rating Curve= 0 ,0
Exp/Cntr(USF)=0,0
Exp/Cntr=0.3,0.1

Type RM Length L Ch R = 1 ,13588   ,330.8,311,267.9
XS GIS Cut Line= 4
2045280.79899722249571.1599853792044684.44131795249563.415080454
2044370.77266846249542.1165919082043985.01613371250008.674132667
#Sta/Elev= 30
       01710.557  22.4151707.158  83.7221692.618 156.0251683.852 195.3991676.893
 513.6661660.354 552.4461661.651 668.0371660.049 684.4791658.861  743.671659.942
 760.1121658.297 766.6891656.186   779.81655.477 798.9931653.872   814.31655.494
 835.7451663.921 849.6271667.228 875.2061678.078 888.3591680.432 910.7991679.886
 963.1921681.5611055.8691683.8981215.4791682.6071283.2241683.3831313.023 1681.09
1341.114 1685.131381.1361688.4551415.6841693.6151469.2811703.1431516.1781713.129
#Mann= 7 ,-1 , 0
       0      .1       0   779.8    .045       0   814.3      .1       0
 910.799      .1       0 963.192      .1       01215.479     .04       0
1341.114      .1       0
#XS Ineff= 2 , 0
             700 1665.83
Permanent Ineff=
       F       F
Bank Sta=779.8,814.3
XS Rating Curve= 0 ,0
Exp/Cntr(USF)=0,0
Exp/Cntr=0.3,0.1

Type RM Length L Ch R = 1 ,13277   ,370.6,360.5,341.3
XS GIS Cut Line= 3
 2044717.3453812  248994.93431892044385.31413117249435.472513318
2043927.41482562249921.583624437
#Sta/Elev= 30
       0 1739.71   105.6 1734.59   189.8    1729   206.5 1727.39   227.1 1723.53
   244.3 1716.94   272.2 1700.49   276.4 1696.51     286  1683.9   302.4 1671.18
   313.3 1656.35   321.1 1652.25   333.9 1650.91   358.6 1652.19   365.6 1652.59
     375 1655.22   391.4 1655.62   402.3 1657.44   445.3 1656.97   465.3 1658.72
   482.8 1661.77   517.9 1672.55     539 1675.47   641.7 1676.89   824.6  1676.2
   961.3 1671.17  1098.5 1671.21  1146.6 1669.16  1173.6 1673.35  1219.5 1676.57
#Mann= 11 ,-1 , 0
       0      .1       0     230      .1       0     240      .1       0
   321.1    .045       0   358.6      .1       0  561.65      .1       0
  611.65      .1       0  751.65      .1       0  881.65      .1       0
 1021.65     .04       0 1151.65      .1       0
#XS Ineff= 2 , 0
                          399.17         1662.22
Permanent Ineff=
       F       F
Bank Sta=321.1,358.6
XS Rating Curve= 0 ,0
Exp/Cntr(USF)=0,0
Exp/Cntr=0.3,0.1

Type RM Length L Ch R = 1 ,12916   ,355.2,352,339.7
XS GIS Cut Line= 4
2044479.20133742248750.2000632622044181.02249778249102.593237379
2044148.10665185249340.7490638422043860.69344558249912.411908514
#Sta/Elev= 30
       0 1769.48    72.5 1758.71   178.9    1747   257.3 1740.89   403.4 1732.97
   454.2 1728.33   473.1 1725.34   486.3 1720.03   496.2 1714.33   512.8 1700.93
   515.9 1697.78     526 1682.83     536 1673.09   545.9 1666.19   549.2  1662.6
   555.9 1652.37  558.411650.747     579 1649.44  608.971650.745   622.1 1653.47
   685.1 1652.84   716.2 1653.93  1083.4 1650.95  1159.4 1652.19  1186.2 1651.34
  1222.9 1653.06  1266.7 1653.64  1311.1 1658.65  1329.5  1662.3  1341.9 1662.73
#Mann= 7 ,-1 , 0
       0     .04       0      60    .035       0     440      .1       0
  558.41    .045       0  608.97      .1       0  752.04    .035       0
 1002.04      .1       0
#XS Ineff= 1 ,-1
  742.13 1278.331661.344
Permanent Ineff=
       T
Bank Sta=558.41,608.97
XS Rating Curve= 0 ,0
Exp/Cntr(USF)=0,0
Exp/Cntr=0.3,0.1

Type RM Length L Ch R = 1 ,12564   ,377.4,369.9,354.8
XS GIS Cut Line= 4
2043969.97383856248616.6004532952043884.77988438249168.424929247
2043847.99158598249439.4966016442043780.68039491  249952.4448842
#Sta/Elev= 30
       0 1751.07   114.8 1731.84   224.4 1715.47   290.7 1709.04   320.6 1708.05
   353.8 1716.39   373.7 1718.76   416.9 1715.73   460.1 1714.92   536.4 1720.84
   556.3 1720.65     563 1719.31   569.6 1716.05   599.4 1681.74   632.5  1653.1
   639.1    1649   672.2 1647.94   688.8 1649.13   738.4 1648.74  757.761646.643
   768.2 1645.37  782.891646.643   794.7 1650.98   844.4  1651.7   988.7 1651.88
    1119 1650.36  1274.5 1652.07    1301 1653.66  1320.9 1656.56  1349.3 1663.88
#Mann= 4 ,-1 , 0
       0      .1       0  757.76    .045       0  782.89    .035       0
  971.92      .1       0
#XS Ineff= 2 , 0
                             900        1657.141
Permanent Ineff=
       F       F
Bank Sta=757.76,782.89
XS Rating Curve= 0 ,0
Exp/Cntr(USF)=0,0
Exp/Cntr=0.3,0.1

Type RM Length L Ch R = 1 ,12194   ,412.3,408,403.3
XS GIS Cut Line= 4
 2043405.0806471248866.8924430782043508.36965503249280.048474776
2043576.24528881249480.7242616012043705.98965748249983.054737402
#Sta/Elev= 30
       0 1699.63    75.4 1699.73     116 1697.86   227.6 1687.36   369.6 1679.21
     400  1678.4   443.1 1665.23   451.4 1660.55   465.2 1655.86   498.5 1649.15
   511.4 1647.48  520.181644.551     531 1642.74   544.6 1642.51   548.3 1642.74
  553.991644.553   562.2 1647.43   579.5 1646.59   586.4 1648.69     607 1649.72
   651.9 1648.22   709.5 1648.51   742.6 1647.78   868.8 1649.44   967.1 1652.18
     991  1651.7  1058.3 1653.61  1112.8 1654.06  1125.7 1655.78  1156.5  1665.3
#Mann= 4 ,-1 , 0
       0    .035       0  435.87      .1       0  520.18    .045       0
  553.99      .1       0
#XS Ineff= 2 , 0
                             607        1651.657
Permanent Ineff=
       F       F
Bank Sta=520.18,553.99
XS Rating Curve= 0 ,0
Exp/Cntr(USF)=0,0
Exp/Cntr=0.3,0.1

Type RM Length L Ch R = 1 ,11786   ,508.1,529.1,523.6
XS GIS Cut Line= 4
2042929.95121065248934.7680768572043068.65359272249356.777452092
2043228.01377637249651.8889033052043381.47173101250023.729331833
#Sta/Elev= 30
       0 1681.53    15.9 1680.01   112.6  1677.8     329 1676.76   437.2  1675.1
   451.6 1671.76   462.6 1667.19     474 1657.74   485.1 1646.15   492.6  1642.2
   545.2 1644.99   585.8 1643.54   607.9 1644.78   656.7 1644.89   663.8  1642.4
     688 1641.14   697.7 1642.72   705.1 1643.93   727.5 1643.82   743.7 1641.77
   753.6 1644.65   779.7 1645.25   818.7 1643.38     840 1643.84   847.9  1642.6
   854.2 1643.53   861.3 1646.44  1127.5 1653.73  1145.3 1657.371181.871 1675.45
#Mann= 5 ,-1 , 0
       0     .04       0      60    .035       0  474.22      .1       0
   663.8    .045       0   697.7      .1       0
#XS Ineff= 2 , 0
                             810            1647
Permanent Ineff=
       F       F
Bank Sta=663.8,697.7
XS Rating Curve= 0 ,0
Exp/Cntr(USF)=0,0
Exp/Cntr=0.3,0.1

Type RM Length L Ch R = 1 ,11257   ,290.9,288.9,286.8
XS GIS Cut Line= 4
2042561.06189663249097.079375024 2042723.3731948249542.697666356
2042782.39548504249802.3957434232042826.66220272250174.236171951
#Sta/Elev= 30
       0 1676.77    63.3 1672.06    93.6 1668.54   112.2 1665.79   143.6 1658.87
   199.5 1653.19   224.6 1653.09   301.2 1656.67   385.3 1651.28   472.4 1651.12
   532.5 1647.97   540.8 1646.05     556 1638.79   569.5 1637.31   581.9 1639.15
   592.9  1637.6     620 1635.97  630.561637.826   636.8 1639.48   650.2 1640.05
   686.1 1638.78     708  1639.8   770.4 1638.63   780.7  1639.9   880.1 1640.98
   952.5 1652.68   992.2 1662.85  1021.9 1674.79  1074.8 1701.971115.045 1726.25
#Mann= 5 ,-1 , 0
       0      .1       0     150    .035       0  514.26      .1       0
   592.9    .045       0  630.56      .1       0
#XS Ineff= 2 , 0
                             810            1644
Permanent Ineff=
       F       F
Bank Sta=592.9,630.56
XS Rating Curve= 0 ,0
Exp/Cntr(USF)=0,0
Exp/Cntr=0.3,0.1

Type RM Length L Ch R = 1 ,10968   ,324.9,342,360.6
XS GIS Cut Line= 4
2042457.77288871 249147.248321732042457.77288871249672.546704889
2042522.69740798249882.0758352512042572.86635468250165.382828415
#Sta/Elev= 30
       0 1676.25    45.4 1672.19    65.1 1669.46    91.3  1662.3   104.5 1656.78
   120.9  1652.2   166.5  1645.9   219.3 1642.24   252.1 1638.71     341 1638.19
   419.4 1639.04     511 1637.69   558.4 1638.55   589.6 1637.24   641.2 1637.62
  647.671635.149   678.9 1633.62  686.32 1635.15   692.7 1638.08   715.8 1636.23
   723.6 1635.44   736.7 1637.73   807.5 1639.94     821 1641.21   837.5 1645.98
   874.8 1665.16   930.8 1704.36   957.4  1720.7   996.5 1741.33 1032.37 1756.83
#Mann= 5 ,-1 , 0
       0      .1       0     341    .035       0  647.67    .045       0
  686.32    .035       0   715.8      .1       0
#XS Ineff= 2 , 0
             560    1642
Permanent Ineff=
       F       F
Bank Sta=647.67,686.32
XS Rating Curve= 0 ,0
Exp/Cntr(USF)=0,0
Exp/Cntr=0.3,0.1

Type RM Length L Ch R = 1 ,10626   ,218.1,216.3,216.3
XS GIS Cut Line= 4
2042369.23945334249182.6616958762042230.53707127249666.644475865
2042121.34583433249926.3425529332042047.56797152250121.116110733
#Sta/Elev= 30
       0 1666.69    44.5 1659.14   103.9 1645.68   144.2 1640.18     168 1639.54
     181 1638.22   239.5 1636.87   286.8 1637.41   411.6  1636.1   460.9 1637.12
   530.3 1633.75   548.1 1633.72     587 1635.84     605 1633.42   637.2 1635.12
  651.461631.543   664.7 1629.69   672.6 1629.95  679.251631.544   683.3 1633.78
   686.9 1637.31     694  1649.8   697.5 1653.26   761.6 1691.62   793.5 1715.42
   833.3 1741.79   891.9 1777.91   916.3  1796.3   954.9 1822.59993.4635 1844.12
#Mann= 6 ,-1 , 0
       0     .04       0      10      .1       0     200    .035       0
  543.47      .1       0  651.46    .045       0  679.25      .1       0
#XS Ineff= 2 , 0
             520    1650
Permanent Ineff=
       F       F
Bank Sta=651.46,679.25
XS Rating Curve= 0 ,0
Exp/Cntr(USF)=0,0
Exp/Cntr=0.3,0.1

Type RM Length L Ch R = 1 ,10410   ,207.6,205.3,200.6
XS GIS Cut Line= 4
 2042260.0482164249144.297207218 2042065.2746586249536.795437332
2041923.62116201249843.7113465932041876.40332982250053.240476954
#Sta/Elev= 30
       0 1671.44      10 1668.47    50.3 1661.59   119.9 1650.66   182.2 1644.18
   215.1  1639.5   270.1 1636.19   324.5 1634.93   390.6 1635.84   498.9  1632.3
   532.5 1632.29   558.2 1634.02  575.761630.368   583.1  1628.9   610.2 1628.98
  617.091630.366   630.1 1636.57   651.7 1657.73   666.2 1669.15   684.3 1681.27
   707.9 1694.57   718.9 1698.92   753.6 1708.16   841.6 1749.65   865.5 1758.19
   875.6 1760.41   889.1 1768.19   937.7 1781.74   978.9 1799.44990.9803 1806.49
#Mann= 6 ,-1 , 0
       0     .04       0    50.3      .1       0   270.1    .035       0
   498.9      .1       0  575.76    .045       0  617.09      .1       0
#XS Ineff= 2 , 0
             500    1650
Permanent Ineff=
       F       F
Bank Sta=575.76,617.09
XS Rating Curve= 0 ,0
Exp/Cntr(USF)=0,0
Exp/Cntr=0.3,0.1

Type RM Length L Ch R = 1 ,10205   ,209.7,201,188.4
XS GIS Cut Line= 4
2041826.23438311249079.3726879512041870.50110079 249409.89751331
2041784.91877994249713.8623080592041781.96766543250000.120415736
#Sta/Elev= 30
       0 1754.07    34.9 1735.31      58 1719.48    71.3 1713.21    87.8  1701.4
   127.5 1678.47   139.9 1669.34   160.4 1668.33   170.6 1661.48   177.9 1658.53
   240.1 1640.29   266.6  1634.8     293 1633.36   482.1 1631.66  490.991628.362
   513.4 1627.17  521.571628.361   530.4 1634.18   540.7  1637.5   557.7 1630.16
   595.2 1631.77   646.3 1660.83   691.9 1689.69   731.7 1697.62   748.1  1705.4
   815.5 1729.22   866.3 1751.36   879.4 1758.71   928.6 1774.65935.5323 1778.53
#Mann= 7 ,-1 , 0
       0      .1       0     110     .04       0     210      .1       0
  413.48    .035       0  490.99    .045       0  521.57    .035       0
  613.48      .1       0
#XS Ineff= 2 , 0
             400    1640     540            1640
Permanent Ineff=
       F       F
Bank Sta=490.99,521.57
XS Rating Curve= 0 ,0
Exp/Cntr(USF)=0,0
Exp/Cntr=0.3,0.1

Type RM Length L Ch R = 1 ,10004   ,205.4,200.8,191.7
XS GIS Cut Line= 4
2041528.17181739249250.5373296552041643.26528336249427.604200383
2041669.82531397249672.5467048892041731.79871872249997.169301224
#Sta/Elev= 30
       0  1743.8    28.8 1732.47    60.1  1716.9    98.7 1690.46   103.4 1686.36
   110.5 1677.52   114.9 1674.51   134.4 1672.62   157.9 1657.66   172.2 1650.94
   200.2 1643.46   238.9  1636.8  257.761627.688   265.3 1625.36   278.6 1625.35
   285.1 1625.67  290.721627.688   311.1 1633.92   331.3  1630.2   354.4 1628.89
   417.1 1629.33   436.9 1631.58   496.7 1653.88   556.9  1671.9   566.9 1679.44
   580.2 1685.43   610.3 1697.75   657.1 1714.65   760.6 1756.39788.0488 1768.88
#Mann= 6 ,-1 , 0
       0      .1       0      40     .04       0  257.76    .045       0
  290.72      .1       0  361.19    .035       0  467.56      .1       0
#XS Ineff= 2 , 0
                           307.2            1640
Permanent Ineff=
       F       F
Bank Sta=257.76,290.72
XS Rating Curve= 0 ,0
Exp/Cntr(USF)=0,0
Exp/Cntr=0.3,0.1

Type RM Length L Ch R = 1 ,9803    ,242.6,235.6,224.4
XS GIS Cut Line= 4
2041377.66497727249330.2174214822041436.68726751249483.675376113
2041522.26958836249705.0089645232041646.21639787249994.218186712
#Sta/Elev= 30
       0 1744.65    63.5 1714.18    81.1 1711.93    91.6 1706.65     102 1703.39
   152.8 1690.73   172.5 1680.53   186.6 1681.12     196 1679.48   214.7 1663.66
   232.3 1636.76  242.671627.481   249.9 1625.04     271 1624.62     278 1625.63
   283.9 1628.42   292.1 1634.55   302.6 1628.98   317.7 1627.34   422.5 1632.29
   465.4 1636.44   483.2 1634.98   504.6 1636.18   511.8 1638.75   522.5 1645.26
   541.4 1650.36   597.5  1672.2   625.3 1684.49   661.7 1703.36716.3707 1735.39
#Mann= 5 ,-1 , 0
       0      .1       0     150     .04       0  242.67    .045       0
   283.9    .035       0  591.72      .1       0
#XS Ineff= 2 , 0
                             300         1643.61
Permanent Ineff=
       F       F
Bank Sta=242.67,283.9
XS Rating Curve= 0 ,0
Exp/Cntr(USF)=0,0
Exp/Cntr=0.3,0.1

Type RM Length L Ch R = 1 ,9567    ,212,215.1,217.3
XS GIS Cut Line= 4
2041032.38457935249424.6530858712041224.20702264249634.182216232
  2041433.736153249849.6135756172041590.14522214250085.702736588
#Sta/Elev= 30
       0 1705.92    26.1  1699.1    69.8 1693.53   112.5 1685.33   148.1 1682.55
   170.3 1677.92   201.4 1677.28   210.3 1675.46   223.7 1668.45   241.5 1667.59
   268.6 1662.26   299.7 1660.28   304.3  1658.4   313.5  1650.4   327.2 1642.54
   338.2  1633.7  354.041626.471   361.4 1624.59   370.7 1626.62   386.9 1630.26
     405 1625.76   501.1 1630.33   551.5  1630.5   570.6 1633.21   608.6 1633.83
   638.6 1636.28   671.7 1643.46   713.5 1661.54   759.3 1685.72867.7953 1753.62
#Mann= 7 ,-1 , 0
       0      .1       0     210     .06       0  344.07      .1       0
  354.04    .045       0   370.7      .1       0  444.07    .035       0
   614.6      .1       0
Bank Sta=354.04,370.7
XS Rating Curve= 0 ,0
Exp/Cntr(USF)=0,0
Exp/Cntr=0.3,0.1

Type RM Length L Ch R = 1 ,9352    ,130.1,133.5,136.7
XS GIS Cut Line= 4
2040938.07939619249456.9463421022041072.73734741249759.291553344
2041216.28780485249951.1156159382041373.81220063250198.835431871
#Sta/Elev= 30
       0 1699.08    59.1 1686.46   116.5 1681.64   140.5 1675.57   148.8 1671.07
   191.9 1671.02   241.8 1664.77   274.6 1655.62   284.7 1650.65     300  1639.7
   321.2 1635.42   332.2 1629.99   364.9 1627.85   385.4 1630.16  396.081623.849
   402.1 1622.07   418.2 1621.88  428.861623.845   437.3 1626.07   481.1 1626.72
   505.3 1629.86   611.3 1631.35     636 1632.61   686.5 1640.69   699.2 1649.09
   725.4 1660.99     742 1671.52   772.9 1694.35     817 1731.73864.1287 1766.34
#Mann= 7 ,-1 , 0
       0      .1       0   140.5     .04       0   241.8      .1       0
  396.08    .045       0  428.86      .1       0   481.1    .035       0
   611.3      .1       0
Bank Sta=396.08,428.86
XS Rating Curve= 0 ,0
Exp/Cntr(USF)=0,0
Exp/Cntr=0.3,0.1

Type RM Length L Ch R = 1 ,9219    ,142.7,153.1,170.8
XS GIS Cut Line= 4
2040935.14128213 249474.798526432041004.92414333249882.759868777
2041129.72810661250106.8702114482041243.79624509250306.824948322
#Sta/Elev= 30
       0 1695.03   125.1 1673.63   139.3 1668.24   186.4 1667.71     223 1654.17
   236.3 1645.97     253 1644.47   289.6 1627.66   386.6 1626.27   406.5 1629.76
   417.2 1629.84   420.1 1629.48   430.2 1622.15   438.9 1620.66   453.4 1621.92
   465.5  1626.1   495.2 1624.36   615.4 1630.15   631.9 1633.23   646.4 1638.55
     683 1640.54   690.6 1644.45   701.9 1656.26     721  1670.3   758.6 1695.77
   769.9 1706.15   811.5 1739.34     853 1769.59   883.2 1787.15   900.6 1793.99
#Mann= 7 ,-1 , 0
       0      .1       0     110     .04       0     210      .1       0
     310     .03       0   430.2    .045       0   453.4     .03       0
  483.89      .1       0
Bank Sta=430.2,453.4
XS Rating Curve= 0 ,0
Exp/Cntr(USF)=0,0
Exp/Cntr=0.5,0.3

Type RM Length L Ch R = 1 ,9065    ,22.8,23.3,25.5
XS GIS Cut Line= 4
2040922.83509982249476.0017125582040905.25148627249958.637064688
2040900.52120575250109.7606170082040972.85414427250442.103835347
#Sta/Elev= 30
       01695.032  84.1651679.603 136.6941671.409 153.109  1665.4 183.3381665.914
 195.7881658.638 212.2031657.108 238.4671647.731  274.581633.016 284.4291627.368
 294.2781625.459 448.5791623.783 464.9951624.927 487.9751629.006 504.3871629.752
 510.9521628.199  518.991621.947 537.2111620.383  542.841622.771 547.0591626.894
 553.6241629.523 586.4481629.747 642.4961637.016 733.091 1676.13 770.0251688.791
  833.821718.736 880.8271735.255 904.4571740.633 931.192 1743.83 974.2771743.258
#Mann= 8 ,-1 , 0
       0      .1       0  84.165     .04       0 183.338      .1       0
 238.467     .06       0 294.278     .03       0 464.995      .1       0
  518.99    .045       0  542.84      .1       0
#XS Ineff= 1 ,-1
205.8265484.2402 1632.43
Permanent Ineff=
       T
Bank Sta=518.99,542.84
XS Rating Curve= 0 ,0
Exp/Cntr(USF)=0,0
Exp/Cntr=0.5,0.3

Type RM Length L Ch R = 1 ,9042    ,118.8,122.8,131.8
XS GIS Cut Line= 4
2040918.25804891249474.3926773612040883.31212192249959.356562039
2040872.61438917250129.0939216762040943.21942532 250447.17317545
#Sta/Elev= 30
       0 1695.55   138.6 1671.49   158.3 1664.65   181.3 1665.59   194.5 1659.63
   210.9 1658.28   247.1 1645.02   260.3 1636.07   270.4 1633.54   291.4 1624.69
   424.7 1625.31     451 1622.68   503.7 1629.64   510.3 1627.93   515.6  1622.4
   520.1 1620.49   543.1  1620.3     553 1622.14   569.4 1628.59   681.7 1638.78
   735.5 1645.99   763.3 1646.77   772.5 1650.67   802.7 1672.33   836.3 1691.23
   873.3 1708.38   893.5 1714.86     917 1719.51     964 1723.77   982.1 1723.42
#Mann= 8 ,-1 , 0
       0      .1       0     110     .04       0     210      .1       0
     300     .06       0     400     .03       0  506.22      .1       0
   515.6    .045       0     553      .1       0
#XS Ineff= 2 , 0
           497.4 1633.57
Permanent Ineff=
       F       F
Bank Sta=515.6,553
XS Rating Curve= 0 ,0
Exp/Cntr(USF)=0,0
Exp/Cntr=0.5,0.3

Type RM Length L Ch R = 1 ,8919    ,143.2,176.6,196.5
XS GIS Cut Line= 4
2040897.42793921249462.0277742232040778.01428435249915.545591086
2040719.57781495250122.6139500462040657.33027146250380.496630223
#Sta/Elev= 30
       0 1699.38   164.9 1669.66   176.1 1661.59   199.9 1661.95     232 1646.81
   237.1 1641.41   243.9 1628.73   245.4  1627.7   264.2 1623.31   338.9 1623.61
   410.2  1621.6   430.5 1623.78     461 1623.41   481.5 1627.46     487 1625.99
   492.9 1621.81   498.5 1619.83   515.6 1618.66   546.2 1619.04   554.8 1621.76
   573.5 1624.51     591 1623.86   607.6 1625.98   631.5 1633.32   641.7 1639.11
   665.1 1643.21   679.2 1654.15   763.6 1692.04   868.2 1733.42949.4205 1759.59
#Mann= 7 ,-1 , 0
       0      .1       0     120     .04       0     230      .1       0
     330     .03       0     430      .1       0   492.9    .045       0
   554.8      .1       0
#XS Ineff= 1 ,-1
208.1354475.4777 1632.43
Permanent Ineff=
       T
Bank Sta=492.9,554.8
XS Rating Curve= 0 ,0
Exp/Cntr(USF)=0,0
Exp/Cntr=0.3,0.1

Type RM Length L Ch R = 1 ,8743    ,161.5,156,152.2
XS GIS Cut Line= 4
2040882.18364285249463.2981322542040723.38888905249820.268738804
2040619.21953055249873.6237760822040365.14792447 250045.12211019
#Sta/Elev= 30
       0 1700.28    55.6 1689.43   100.3 1677.49   138.3 1670.38   152.5 1666.17
   163.4 1658.57   187.3 1658.38   200.6 1650.06   217.3 1643.58   222.1  1640.7
     228 1634.78   235.2  1624.1   238.8 1622.75   249.6 1621.83   303.5 1622.69
   378.7 1620.45   421.8 1621.53  442.64 1617.82   458.7 1616.38   471.5 1617.82
   480.8  1623.9   493.5 1626.12   510.4 1633.52   550.1 1647.46   626.2  1679.5
   656.9 1695.18   686.2 1714.23   721.4 1734.26   787.6 1761.68814.2706 1778.05
#Mann= 9 ,-1 , 0
       0      .1       0     110     .04       0     240      .1       0
     340    .035       0     350      .1       0  442.64    .045       0
   471.5      .1       0   490.7    .035       0  507.74      .1       0
#XS Ineff= 2 , 0
             400    1633
Permanent Ineff=
       F       F
Bank Sta=442.64,471.5
XS Rating Curve= 0 ,0
Exp/Cntr(USF)=0,0
Exp/Cntr=0.3,0.1

Type RM Length L Ch R = 1 ,8587    ,185.1,178.8,169.7
XS GIS Cut Line= 4
2040868.20970452249454.4056260412040670.03385177249664.014701061
 2040525.2130363249770.7247756172040324.49646749249960.008122151
#Sta/Elev= 30
       0 1703.74    31.5 1697.99    64.2 1689.01   122.6 1666.52   136.5 1660.32
     150 1651.93   171.3 1651.16   185.2  1641.9   199.7 1636.95   227.3  1630.3
   246.4  1623.6   260.7 1621.46   285.4 1619.99   313.7 1620.86   327.2  1619.5
  334.76 1616.54   340.1 1615.12   362.2 1615.15  369.771616.542   378.8 1621.56
   395.3 1622.58   407.4 1632.54   428.1 1641.82   495.9 1668.83   542.3 1693.68
   590.3 1724.69   639.9 1753.26   700.1 1783.72   721.1 1792.52  744.24 1799.44
#Mann= 7 ,-1 , 0
       0      .1       0      50     .04       0     190      .1       0
  308.46    .035       0  334.76    .045       0  369.77    .035       0
  448.46      .1       0
#XS Ineff= 2 , 0
             300    1625     380            1625
Permanent Ineff=
       F       F
Bank Sta=334.76,369.77
XS Rating Curve= 0 ,0
Exp/Cntr(USF)=0,0
Exp/Cntr=0.3,0.1

Type RM Length L Ch R = 1 ,8408    ,130.5,134.5,137.4
XS GIS Cut Line= 4
2040747.52569162249298.1515882982040600.16416009 249450.59455195
2040489.64301145249615.7410959052040296.54859082249891.408788508
#Sta/Elev= 30
       0 1735.26    43.3 1718.75    76.9 1701.11   138.4 1665.83   173.8 1650.53
   189.5 1642.13   217.5 1641.21   233.3 1638.37   245.1  1633.5   258.6 1630.71
   293.1 1627.68   300.4 1624.91  311.931615.378   316.2 1613.66   323.8  1613.5
  340.321615.374   382.5 1616.89   394.3 1623.35   406.1 1626.07   410.9 1629.01
   418.9 1637.81   426.9 1643.58   477.3 1668.91     491 1677.64   503.4  1682.3
   520.6 1692.07   591.2 1722.77   695.3 1781.94   719.9 1792.35747.3091 1801.34
#Mann= 5 ,-1 , 0
       0      .1       0     120     .06       0     160     .04       0
  311.93    .045       0  340.32      .1       0
Bank Sta=311.93,340.32
XS Rating Curve= 0 ,0
Exp/Cntr(USF)=0,0
Exp/Cntr=0.3,0.1

Type RM Length L Ch R = 1 ,8273    ,253.4,256.1,257
XS GIS Cut Line= 4
2040666.22277768249216.8486743512040485.83193736249401.050588763
2040352.44434416249552.2231943842040227.94925718249714.829022279
#Sta/Elev= 30
       0 1740.54    67.2 1707.59   117.7 1676.08   136.1 1663.39   168.9 1648.84
   192.4 1640.44   215.8  1640.3   229.9 1633.64   238.2 1631.58   259.9 1627.83
   298.6 1623.68  319.26 1614.06   333.4 1612.94   356.41614.061   369.3 1616.39
   386.8 1627.44   401.8 1628.24   408.7 1630.58   421.7 1641.89   426.6 1649.08
     431 1653.28   531.3 1725.86   561.9 1746.78   574.9    1754   576.8 1755.77
   585.6 1769.39   605.7 1779.51   627.4 1787.62     645 1792.36664.2189 1795.58
#Mann= 4 ,-1 , 0
       0      .1       0     180     .04       0  319.26    .045       0
   356.4      .1       0
Bank Sta=319.26,356.4
XS Rating Curve= 0 ,0
Exp/Cntr(USF)=0,0
Exp/Cntr=0.3,0.1

Type RM Length L Ch R = 1 ,8017    ,176.1,174.7,163.5
XS GIS Cut Line= 4
2040506.15766584249018.6728216042040329.57789961249211.767242229
2040225.40854112249315.9366007242040097.10238005249534.438181958
#Sta/Elev= 30
       0 1751.19    28.5 1737.25    71.3 1712.41   102.4 1691.07   121.4 1681.02
   142.3 1672.61   210.2 1649.96   225.9 1640.03   244.5 1639.71   256.1  1637.6
   283.9 1618.84  299.121611.448     310 1610.03  335.991611.449   350.6 1616.66
   398.2 1620.85   413.3 1629.02   433.4 1633.08   448.6 1633.37   473.9 1638.96
   481.1 1641.83   493.1 1650.21   498.1 1652.27   528.5    1654   535.8 1659.28
   545.8 1669.37   562.6 1679.31   588.2  1698.6   627.3 1725.45662.3654 1746.37
#Mann= 5 ,-1 , 0
       0      .1       0      90     .04       0     240      .1       0
  299.12    .045       0  335.99      .1       0
Bank Sta=299.12,335.99
XS Rating Curve= 0 ,0
Exp/Cntr(USF)=0,0
Exp/Cntr=0.3,0.1

Type RM Length L Ch R = 1 ,7843    ,107.2,104.1,100.8
XS GIS Cut Line= 4
2040377.85150477248894.1777346222040213.97531884249070.757500852
2040111.07631838249230.8226126862040020.88089822249432.809539524
#Sta/Elev= 30
       0 1724.25    26.8 1714.25    58.3  1699.7   111.6 1678.31   150.1  1659.2
   178.9 1646.25   201.3 1638.51   216.2 1634.38   225.4 1630.03   241.5 1629.93
   251.2 1628.63   263.1 1621.49   276.6 1617.35  290.571608.745   296.1 1607.66
  329.441608.746   331.9  1609.8     339 1615.49   342.9 1616.52   369.9 1619.03
   403.1 1624.83   424.8 1626.77   504.4 1641.51   540.3 1650.06   553.4 1652.02
   570.8 1659.27   594.2 1661.84   615.8 1667.35   630.4 1672.85652.4031 1684.27
#Mann= 5 ,-1 , 0
       0      .1       0     130     .04       0  260.91      .1       0
  290.57    .045       0  329.44      .1       0
Bank Sta=290.57,329.44
XS Rating Curve= 0 ,0
Exp/Cntr(USF)=0,0
Exp/Cntr=0.3,0.1

Type RM Length L Ch R = 1 ,7738    ,102.8,107,112.7
XS GIS Cut Line= 4
2040229.21961521248812.8748206752040118.69846656249009.780315391
2040048.82877489249164.7639951032040001.82552776249412.483811037
#Sta/Elev= 30
       0 1689.59    25.7 1679.49    85.6 1651.79    93.1 1649.54   114.7 1646.44
   143.6 1637.92   170.1 1631.88   213.5 1623.59   239.3 1623.89   250.1 1619.23
   260.2 1612.73   264.5 1612.04   272.6 1609.03   280.1  1606.2   289.6  1605.5
   298.8 1606.07   309.8 1609.34   319.8  1614.8   346.7 1619.39     358 1625.62
   366.9  1628.4   420.9 1633.59   484.3 1646.34     511 1647.58   530.4 1650.22
   561.1  1657.6   587.8 1658.29   604.5 1663.72   634.6 1670.32647.9471 1674.62
#Mann= 5 ,-1 , 0
       0      .1       0   170.1     .04       0   264.5      .1       0
   272.6    .045       0   309.8      .1       0
Bank Sta=272.6,309.8
XS Rating Curve= 0 ,0
Exp/Cntr(USF)=0,0
Exp/Cntr=0.3,0.1

Type RM Length L Ch R = 1 ,7631    ,154,154.3,160.5
XS GIS Cut Line= 4
2040160.74820717248792.8166657252040043.08765303248952.277679889
2039953.29407223249079.2272251462039858.85599588249221.658422263
#Sta/Elev= 30
       0 1654.78    11.7 1651.08    44.2 1637.51    53.6 1634.81    93.3 1627.74
   113.6 1626.17     134  1625.4   182.1 1620.02   194.3 1620.88   206.1 1620.55
   210.8 1619.02   221.4 1613.12   224.9 1612.33   232.8 1612.25   238.5 1611.45
   250.8 1605.65   279.1 1604.64   291.7 1605.57   295.7 1606.79   299.7 1609.57
   307.8 1616.67   323.7 1617.52   329.4 1618.59   368.6 1630.55   399.5 1642.04
   429.2 1656.57   458.5 1673.08   482.2 1685.73   505.5 1696.52   524.6 1703.44
#Mann= 4 ,-1 , 0
       0      .1       0     120     .04       0   250.8    .045       0
   291.7      .1       0
Bank Sta=250.8,291.7
XS Rating Curve= 0 ,0
Exp/Cntr(USF)=0,0
Exp/Cntr=0.3,0.1
